--- LaurelCrk5.prj (project) ---

Proj Title=LaurelCrk5
Current Plan=p01
Default Exp/Contr=0,0
English Units
Geom File=g01
Flow File=f01
Plan File=p01
BEGIN DESCRIPTION:
END DESCRIPTION:
DSS Export Rating Curves= 0
DSS Export Rating Curve Sorted= 0
DSS Export Volume Flow Curves= 0
DXF OffsetX= 0
DXF OffsetY= 0
DXF ScaleX= 0
DXF ScaleY= 0

--- LaurelCrk5.p01 (plan) ---

Plan Title=Floodplain
Program Version=4.00
Geom File=g01
Flow File=f01
K Sum by GR=0
Std Step Tol=0.01
Critical Tol=0.01
Num of Std Step Trials=20
Max Error Tol=0.3
Flow Tol Ratio=0.001
Split Flow NTrial=30
Split Flow Tol=0.02
Split Flow Ratio=0.02
Log Output Level=0
Friction Slope Method=1
Unsteady Friction Slope Method=2
Unsteady Bridges Friction Slope Method=1
Global Log Level=0
CheckData=False
Run HTab=0
Run UNet=0
Run PostProcess=0
UNET Theta=0
UNET Theta Warmup=0
UNET ZTol=0
UNET ZSATol=0
UNET MxIter=0
UNET MaxInSteps=0
UNET DtIC=0
UNET DtMin=0
UNET MaxCRTS=0
UNET WFStab=0
UNET SFStab=0
UNET WFX=0
UNET SFX=0
UNET DSS MLevel=0
UNET DZMax Abort=0
UNET Convert EG Bridges=0
UNET Use Existing IB Tables=0
UNET Froude Limit=0
UNET Froude Power=0
Write IC File=0
Echo Input=False
Echo Output=False
Write Detailed=0

--- LaurelCrk5.f01 (steady flow) ---

Flow Title=NFF Regression Equation
Program Version=4.00
Number of Profiles=1
Profile Names=P100yr
River Rch & RM=LaurelCrk5,Main      ,19857.8
540.5761
River Rch & RM=LaurelCrk5,Main      ,16450.9
590.5582
River Rch & RM=LaurelCrk5,Main      ,12833.9
655.4587
River Rch & RM=LaurelCrk5,Main      ,12539.8
772.3794
River Rch & RM=LaurelCrk5,Main      ,10165.7
806.3964
River Rch & RM=LaurelCrk5,Main      ,9735.1
1518.821
River Rch & RM=LaurelCrk5,Main      ,7171.1
1616.156
River Rch & RM=LaurelCrk5,Main      ,278.8
1788.054
Boundary for River Rch & Prof#=LaurelCrk5,Main      ,1
Up Type=0
Dn Type=3
Dn Slope=0.016709

--- LaurelCrk5.g01 (geometry) ---

Geom Title=USGS 3m DEM
Program Version=4.10

River Reach=LaurelCrk5      ,Main
Reach XY= 30
     2005881.993       367704.28     2006072.965      368468.169
     2006241.368      368490.738     2006099.006      368898.724
     2006399.354      369428.238     2006295.187      369747.682
     2006365.955      370369.182     2006164.979      370622.682
     2006361.607      371234.804     2006550.395      371662.613
     2006987.895      371841.433     2008005.604      372962.382
     2009195.874      372443.682     2009328.488      372185.183
     2010152.826       372204.28     2010270.926      372051.002
     2010542.667      372061.505     2011225.743      372659.141
     2011750.048      372825.808      2012088.59      373518.516
     2012497.901        373978.3     2012796.389      373928.238
     2013277.231      374264.746     2014093.798      374374.419
     2014500.135      374692.486     2014887.201       374641.78
     2015225.902      375161.937     2016597.271      376565.391
     2016958.381      376657.405     2017949.064      377370.757

Type RM Length L Ch R = 1 ,19857.8 ,557.1,555.8,547.2
XS GIS Cut Line= 3
     2005398.787      368140.507     2005967.392      367935.246
     2006178.446      367898.001
#Sta/Elev= 30
       0 2630.65    19.8 2624.98    39.6 2620.15    59.5 2616.34    79.3 2613.43
   178.4  2603.2   188.3 2602.46   208.1 2603.01     218 2602.67   247.8 2600.34
   277.5 2597.26   307.2 2593.16     337 2587.98   346.9 2585.83   396.4 2571.76
   416.2 2567.11   515.3 2552.54   530.4 2551.08   535.2 2550.84   545.4 2551.23
   604.5 2559.44   614.3 2561.53   633.7 2568.12   672.7 2584.22   692.2 2590.37
   711.7  2594.9   740.9 2599.69   770.1 2603.26   789.6 2604.96   818.8 2606.48
#Mann= 3 , 0 , 0
       0      .1       0   530.4    .045       0   545.4      .1       0
Bank Sta=530.4,545.4
XS Rating Curve= 0 ,0
Exp/Cntr=0.3,0.1

Type RM Length L Ch R = 1 ,19301.2 ,433.2,456.5,465
XS GIS Cut Line= 3
     2005743.923      368384.667     2005945.045      368374.735
      2006439.16      368168.647
#Sta/Elev= 30
       0 2615.17    28.8  2613.4    38.4 2611.96    47.9 2609.75    86.3 2599.04
   115.1 2589.33     163 2574.14   201.4 2561.04   221.2 2557.38   280.7 2549.06
   289.6 2548.34   300.5 2548.12   304.6 2548.13   320.3 2548.46   340.2 2550.61
     360 2554.48   389.7 2561.79   429.4 2574.02     479 2591.95   508.7 2600.67
   528.5 2608.04   538.4 2610.58   548.4  2610.7   568.2 2609.66   627.7 2609.98
   637.6 2610.34   647.5 2611.56   667.3 2615.47   687.2  2620.2   736.7  2635.1
#Mann= 3 , 0 , 0
       0      .1       0   289.6    .045       0   304.6      .1       0
Bank Sta=289.6,304.6
XS Rating Curve= 0 ,0
Exp/Cntr=0.3,0.1

Type RM Length L Ch R = 1 ,18844.1 ,288.2,285.5,282.7
XS GIS Cut Line= 3
     2005572.634      368636.395     2006228.106      368603.171
     2006367.153      368565.926
#Sta/Elev= 30
       0 2664.95    29.8 2655.13    49.7 2649.25    69.6 2643.79    89.5 2639.05
   119.3 2633.87     179 2626.49   198.9 2623.57   218.8 2619.41   288.4 2599.79
   298.3 2595.74   318.2 2585.86   328.2 2582.09   338.1 2579.16     358  2574.7
   427.6 2564.15   517.1 2553.51   556.9  2550.1   616.5 2547.52   624.3 2546.57
   636.4 2545.59   639.3 2546.06   646.4  2547.2   656.3 2549.86   665.9 2551.62
   704.3 2556.45   713.9    2558   723.5 2560.31   733.1 2563.45   800.3 2588.62
#Mann= 3 , 0 , 0
       0      .1       0   624.3    .045       0   639.3      .1       0
Bank Sta=624.3,639.3
XS Rating Curve= 0 ,0
Exp/Cntr=0.3,0.1

Type RM Length L Ch R = 1 ,18558.6 ,154.1,142.6,131.1
XS GIS Cut Line= 2
     2005627.222      368923.476     2006501.235       368776.98
#Sta/Elev= 30
       0 2662.54    19.9 2653.78    79.7 2633.92    99.6 2628.69   119.5 2625.44
   129.4 2624.45   169.3  2623.1   179.2 2621.89   268.8 2599.95   288.8 2597.58
   338.6 2593.86   348.5 2591.52   358.5 2587.48   378.4 2577.13   428.2 2547.73
   438.1 2542.31   448.1 2539.85     458 2539.69   458.5  2539.7   473.5 2539.87
   527.7 2540.75   587.5 2543.02   657.2  2547.1   716.9 2551.39   726.9 2553.23
   736.8 2556.13   836.4 2589.97   846.4 2592.71   866.3    2597   886.2 2603.94
#Mann= 3 , 0 , 0
       0      .1       0   458.5    .045       0   473.5      .1       0
Bank Sta=458.5,473.5
XS Rating Curve= 0 ,0
Exp/Cntr=0.3,0.1

Type RM Length L Ch R = 1 ,18415.8 ,82.4,89.5,99.3
XS GIS Cut Line= 5
     2005886.144       369037.45     2006101.323      369006.151
     2006183.483      368941.598     2006361.495      368884.868
     2006574.718      368832.052
#Sta/Elev= 30
       0 2598.95     9.9 2597.57    19.8 2596.65    69.2 2592.86    79.1 2591.22
      89 2588.26    98.8 2584.57   118.6 2576.53   158.1 2559.77   177.9 2552.32
   187.8 2549.07   207.6 2543.63   217.4 2541.42   236.4 2538.69   245.9 2537.86
   251.9 2537.67   255.4 2537.56   266.9 2537.89   361.3 2541.07   420.3 2543.45
   498.9 2547.35   508.8  2548.6   518.8 2551.17   528.7 2554.68   628.6  2591.3
   638.6 2593.71   648.6 2595.26   658.5 2597.86   718.4 2619.42   728.4 2621.72
#Mann= 3 , 0 , 0
       0      .1       0   251.9    .045       0   266.9      .1       0
Bank Sta=251.9,266.9
XS Rating Curve= 0 ,0
Exp/Cntr=0.3,0.1

Type RM Length L Ch R = 1 ,18326.4 ,296.2,298.9,299
XS GIS Cut Line= 3
     2005660.527      369255.766     2006166.053      369063.736
     2006725.784      368926.994
#Sta/Elev= 30
       0 2656.17    60.1 2646.43    90.1 2640.18   140.2 2627.33   220.3 2603.09
   230.3 2601.46   260.4 2599.78   310.4  2593.3   320.5 2590.53   340.5  2582.2
   390.6 2568.91   430.6 2554.59   460.7 2545.16   480.7 2540.38   510.7 2537.56
   533.3 2533.02   548.3 2533.22   570.6 2533.74   640.1 2531.68   709.6 2535.11
   779.2 2544.54   789.1  2547.7   888.5 2589.08   898.4  2592.3   928.2  2595.4
   948.1 2599.88     968 2607.41   997.8 2620.59  1027.6  2626.6    1117 2649.88
#Mann= 3 , 0 , 0
       0      .1       0   533.3    .045       0   548.3      .1       0
#XS Ineff= 2 , 0
                          585.73         2542.16
Permanent Ineff=
       F       F
Bank Sta=533.3,548.3
XS Rating Curve= 0 ,0
Exp/Cntr=0.3,0.1

Type RM Length L Ch R = 1 ,18027.6 ,136.8,139.5,142.1
XS GIS Cut Line= 4
     2006069.158      369390.406     2006159.386      369363.998
     2006439.976      369289.174     2006497.194      369238.558
#Sta/Elev= 28
       0 2557.61     9.4 2555.97    28.2 2552.52    37.6 2550.57      47 2548.15
    56.4 2545.44    65.8 2542.59    75.2 2539.29      94 2531.45     104 2528.48
     114 2527.47   238.8 2527.42   253.8 2527.42   284.3 2527.38   294.3 2527.08
   304.3 2526.48   334.3  2524.1   344.4 2523.57   354.4 2523.43   364.4 2523.91
   374.4  2525.1   384.4 2526.71     394 2528.65   403.5 2530.81   413.1 2533.11
   422.6 2535.51   441.7 2540.56   460.8 2545.87
#Mann= 3 , 0 , 0
       0      .1       0   238.8    .045       0   253.8      .1       0
#XS Ineff= 2 , 0
          176.65 2531.18
Permanent Ineff=
       F       F
Bank Sta=238.8,253.8
XS Rating Curve= 0 ,0
Exp/Cntr=0.3,0.1

Type RM Length L Ch R = 1 ,17887.9 ,249.9,254.5,259.3
XS GIS Cut Line= 2
     2005832.363      369508.266     2007058.206      369332.547
#Sta/Elev= 30
       0 2613.48      10 2610.32      20 2609.49    49.9  2611.3   109.9 2605.12
   129.8 2598.94   199.7 2565.54   209.7 2562.84   289.6 2547.94   309.6 2545.44
   359.5 2542.35   519.3 2535.45   539.3 2531.84   564.6 2522.49   569.2 2521.08
   579.6 2520.97   619.2 2520.79   639.2 2522.02   669.1 2526.29     739 2544.89
     759 2552.55     789 2569.46   828.9 2586.87   838.9 2589.33   868.9 2592.41
   878.8 2594.45   958.7 2621.56  1018.7 2627.84  1158.5 2650.05  1238.4 2660.08
#Mann= 3 , 0 , 0
       0      .1       0   564.6    .045       0   579.6      .1       0
Bank Sta=564.6,579.6
XS Rating Curve= 0 ,0
Exp/Cntr=0.3,0.1

Type RM Length L Ch R = 1 ,17633.4 ,199.5,200.1,200.2
XS GIS Cut Line= 2
     2005901.943      369626.943     2006895.865      369714.887
#Sta/Elev= 30
       0 2612.31    39.9 2607.55    49.9 2605.46    59.9  2601.6    69.8 2596.38
    99.8 2578.69   129.7 2562.94   149.7 2553.79   159.6 2550.81   209.5 2540.53
   249.4 2536.39   369.2 2519.64   399.1 2516.51   417.7 2515.23   429.1 2515.13
   432.7  2515.2   558.8  2518.7   568.8 2519.87   608.7 2527.65   708.4 2545.66
   728.4 2550.86   738.4 2554.52   818.2 2588.55   828.2 2592.59   838.2 2595.72
   848.1 2596.94     908 2597.44   977.8 2596.27   987.8 2598.17   997.8    2603
#Mann= 3 , 0 , 0
       0      .1       0   417.7    .045       0   432.7      .1       0
Bank Sta=417.7,432.7
XS Rating Curve= 0 ,0
Exp/Cntr=0.3,0.1

Type RM Length L Ch R = 1 ,17432.9 ,358.5,356.2,353.8
XS GIS Cut Line= 2
     2005764.983      369835.101     2006893.485      369838.452
#Sta/Elev= 30
       0 2651.25      20 2640.77      40 2627.02    49.9 2621.11    59.9 2618.02
   169.8 2617.38   189.8 2616.11   209.7    2613   219.7 2609.84   239.7 2600.38
   289.6 2571.48   329.6 2549.16   339.6  2545.1   349.5 2542.64   439.4 2525.74
   479.4    2520   519.3 2516.45   579.2 2514.99     580    2515     595 2515.28
     719 2521.15     789 2530.56   818.9 2535.68   878.8 2549.17   968.7 2582.62
   998.7 2592.03  1018.6 2597.04  1028.6 2598.18  1088.6 2600.54  1128.5 2598.82
#Mann= 3 , 0 , 0
       0      .1       0     580    .045       0     595      .1       0
Bank Sta=580,595
XS Rating Curve= 0 ,0
Exp/Cntr=0.3,0.1

Type RM Length L Ch R = 1 ,17076.2 ,335.7,340.6,345.1
XS GIS Cut Line= 3
     2005935.923      370124.658     2006417.647      370112.665
      2006709.48      370134.652
#Sta/Elev= 30
       0 2607.52    19.7 2598.62      59 2579.89   108.2 2554.52     118 2549.94
   127.8  2545.9   137.7 2542.76   147.5 2540.64   157.4  2539.1   196.7 2533.76
   206.5 2532.16   216.4 2530.14   226.2 2527.71   255.7 2519.74   265.5 2517.89
   275.4 2516.83   324.5 2513.92     342 2513.62     357 2513.62   432.7 2513.76
   442.5 2514.32   452.4 2515.47   511.1 2524.06   569.7 2533.01     638 2542.57
     677 2548.41   706.2 2553.26   725.8 2556.86     755 2562.79   774.5 2567.15
#Mann= 3 , 0 , 0
       0      .1       0     342    .045       0     357      .1       0
Bank Sta=342,357
XS Rating Curve= 0 ,0
Exp/Cntr=0.3,0.1

Type RM Length L Ch R = 1 ,16735   ,272,283.6,293.3
XS GIS Cut Line= 3
     2006129.812      370300.557     2006233.753      370284.566
     2006781.438      370384.509
#Sta/Elev= 30
       0 2536.27    76.5 2527.54      86 2526.01    95.6 2523.86   115.1 2518.99
     125 2516.86     135 2515.21   144.9 2514.21   154.9 2513.77   174.8 2513.62
   187.9 2513.62   202.9 2513.62   244.4 2513.79   254.3 2514.42   264.2 2515.58
   343.8 2526.38   393.5 2532.82   413.4  2536.2   423.3 2538.11   443.2 2542.18
   463.1 2546.58   512.8 2558.44   522.7 2561.06   532.6 2564.61   552.5 2573.84
   582.4  2586.3   602.2 2595.22   622.1 2603.48     642 2610.46   661.9 2616.33
#Mann= 3 , 0 , 0
       0      .1       0   187.9    .045       0   202.9      .1       0
Bank Sta=187.9,202.9
XS Rating Curve= 0 ,0
Exp/Cntr=0.3,0.1

Type RM Length L Ch R = 1 ,16450.9 ,379.6,366.3,349.7
XS GIS Cut Line= 3
     2006085.837      370438.478     2006219.761      370498.444
     2006401.656       370608.38
#Sta/Elev= 30
       0 2536.68     9.8 2535.25    39.1 2531.25    58.7  2528.3    78.3 2524.88
      88    2523    97.8 2520.97   117.4 2516.58   127.2 2514.69     137 2513.78
   139.2 2513.78   146.7 2513.79   154.2 2514.59   156.4 2514.83   166.1 2516.69
   175.7 2518.34   185.4  2519.5     195 2520.25   204.7 2520.83     224  2521.6
   243.3 2521.85     253  2521.7   262.7 2521.38     282 2520.26   291.6 2519.89
   301.3 2519.91     311 2520.27   320.6 2520.94     340  2522.8   359.3 2524.91
#Mann= 3 , 0 , 0
       0      .1       0   139.2    .045       0   154.2      .1       0
Bank Sta=139.2,154.2
XS Rating Curve= 0 ,0
Exp/Cntr=0.3,0.1

Type RM Length L Ch R = 1 ,16084.3 ,186.7,187.3,188.6
XS GIS Cut Line= 3
     2005995.889       370836.25     2006263.735       370784.28
     2006831.301      370683.191
#Sta/Elev= 30
       0 2542.34    29.2 2539.75      78 2532.79   107.2 2527.96   116.9 2526.07
   146.2 2519.59   155.9 2517.75   165.6 2516.49   243.6  2511.2     284  2510.8
     299 2510.77   322.5 2511.05   332.5 2511.85   362.3 2516.33   421.9 2527.08
   451.8 2531.83   531.3 2541.87   541.2 2542.87   590.9 2546.21   610.8 2549.16
   660.5 2558.93   670.4 2561.97   680.4 2566.84   690.3 2573.56   720.1 2597.88
   730.1 2604.85     740 2609.92   749.9 2612.41   759.9 2613.01   849.3 2613.79
#Mann= 3 , 0 , 0
       0      .1       0     284    .045       0     299      .1       0
Bank Sta=284,299
XS Rating Curve= 0 ,0
Exp/Cntr=0.3,0.1

Type RM Length L Ch R = 1 ,15896.7 ,235.1,231.3,226.7
XS GIS Cut Line= 3
     2005769.814      371034.495     2006317.704      370956.181
     2006860.477      370898.434
#Sta/Elev= 30
       0 2560.44    39.5 2554.13   118.6 2544.42   158.1 2540.58   247.1 2537.24
     336 2534.85   355.8 2532.75   375.6 2529.86     425 2520.38   444.7 2517.72
   513.9 2511.62   543.6 2510.05   546.4 2510.13   561.4 2511.34   652.7 2526.56
   712.2 2540.37   761.9 2551.13   801.6 2560.78   841.3 2572.77   851.2  2576.8
   861.1 2582.32     881 2595.14   900.8  2606.1   910.7 2610.46   920.7 2612.97
   930.6 2613.96   990.1 2616.74  1049.7  2618.8  1059.6 2621.25  1099.3 2640.72
#Mann= 3 , 0 , 0
       0      .1       0   546.4    .045       0   561.4      .1       0
Bank Sta=546.4,561.4
XS Rating Curve= 0 ,0
Exp/Cntr=0.3,0.1

Type RM Length L Ch R = 1 ,15665.4 ,381.2,374.1,371.4
XS GIS Cut Line= 2
     2005828.635      371342.473     2006878.717      371015.704
#Sta/Elev= 30
       0 2638.82      70 2635.22      80 2633.58      90 2630.11     120 2615.32
     160 2597.42     190 2586.96     220 2577.72   249.9 2569.36   339.9 2547.11
   409.9 2528.64   439.9 2522.34   469.9 2517.44   489.9 2515.09   546.9 2510.28
   549.9 2510.15   561.9 2511.04   689.8 2532.94   729.8 2541.62   749.8 2547.23
   809.8 2565.31   849.8 2578.75   859.8 2584.04   889.8 2605.03   899.8 2610.64
   909.8 2613.31  1019.8 2619.23  1029.8  2620.3  1039.8  2622.9  1099.8  2645.8
#Mann= 3 , 0 , 0
       0      .1       0   546.9    .045       0   561.9      .1       0
Bank Sta=546.9,561.9
XS Rating Curve= 0 ,0
Exp/Cntr=0.3,0.1

Type RM Length L Ch R = 1 ,15291   ,364.3,359.1,327.5
XS GIS Cut Line= 3
     2006213.764      371705.751     2006497.291      371503.655
     2006623.529      371415.917
#Sta/Elev= 30
       0 2553.92    19.9 2552.65    29.8  2551.9    49.7 2549.91    89.5 2545.51
   119.4 2541.96   129.3 2540.89   139.3 2539.62   159.2 2536.07     199 2527.94
   218.9 2524.08   228.8 2522.29   248.7  2519.4   288.5 2514.64   318.3 2510.56
   328.3 2509.33     337 2508.71   338.2 2508.62   348.2 2508.54     352 2508.56
     377 2508.93   386.6 2509.67   396.2 2511.05   405.8  2512.8   434.7 2518.74
   463.5 2523.73   473.1 2525.86   482.7 2528.47   492.3 2530.39   501.9 2531.74
#Mann= 3 , 0 , 0
       0      .1       0     337    .045       0     352      .1       0
Bank Sta=337,352
XS Rating Curve= 0 ,0
Exp/Cntr=0.3,0.1

Type RM Length L Ch R = 1 ,14930.7 ,325.7,330.1,334.2
XS GIS Cut Line= 2
     2006423.644      372095.528     2006992.595      371202.358
#Sta/Elev= 30
       0 2628.65    69.9 2607.01   179.8 2574.39   219.8 2564.95   319.7 2545.27
   339.7 2539.53   389.6 2522.81   409.6    2517   439.6 2510.63   461.1 2507.47
   469.6 2506.96   476.1 2507.07   519.5 2511.35   629.4 2525.02   699.3 2532.53
   739.3 2538.34   779.3 2545.12   809.2 2551.51   829.2 2556.62   859.2 2565.34
   869.2 2568.93   889.2 2578.68   929.1 2602.92   939.1  2607.8   949.1 2610.84
   959.1 2612.42    1009 2617.49    1039 2617.66    1049 2618.34    1059 2622.04
#Mann= 3 , 0 , 0
       0      .1       0   461.1    .045       0   476.1      .1       0
Bank Sta=461.1,476.1
XS Rating Curve= 0 ,0
Exp/Cntr=0.3,0.1

Type RM Length L Ch R = 1 ,14600.2 ,397.2,398.2,399.2
XS GIS Cut Line= 2
     2006562.129      372241.334     2007137.901      371653.115
#Sta/Elev= 30
       0 2600.92    89.2 2571.25     119 2562.04   148.8 2553.46   168.6 2548.29
   178.5  2546.1   218.2 2538.14   247.9 2532.97   267.8 2530.23   277.7  2529.2
   297.5 2527.78   327.3 2526.42   396.7 2524.13   416.5 2523.15   446.3 2521.06
     476 2518.26   565.3 2507.72   573.9 2507.08   575.2 2506.98   585.1 2507.64
   588.9 2508.59     595 2510.11   614.9  2516.2   674.4 2531.97   684.3 2534.83
   694.2 2538.34   743.8 2560.28   763.6 2568.51   803.3  2584.5   823.1 2592.83
#Mann= 3 , 0 , 0
       0      .1       0   573.9    .045       0   588.9      .1       0
Bank Sta=573.9,588.9
XS Rating Curve= 0 ,0
Exp/Cntr=0.3,0.1

Type RM Length L Ch R = 1 ,14202   ,431.7,423.7,417.5
XS GIS Cut Line= 2
     2006847.213      372471.015     2007377.763      371975.596
#Sta/Elev= 30
       0 2574.53    19.9 2569.65    69.6 2557.03    99.4  2550.1   109.4  2548.1
   119.3 2546.38   139.2 2543.25   159.1 2540.36     179 2538.15   208.8 2535.36
   228.7  2533.1   248.6 2531.33   278.4 2528.35   298.3 2527.18     348 2524.78
     358 2524.01   487.2 2510.77   515.4  2507.6     527    2507   530.4 2507.47
     537 2508.38   546.9 2511.88   556.8 2515.88   616.5 2537.27   636.4  2544.1
   646.3 2547.89   656.3 2552.56   676.2 2562.95   696.1 2573.93   725.9 2590.82
#Mann= 3 , 0 , 0
       0      .1       0   515.4    .045       0   530.4      .1       0
Bank Sta=515.4,530.4
XS Rating Curve= 0 ,0
Exp/Cntr=0.3,0.1

Type RM Length L Ch R = 1 ,13778.3 ,231.1,238.8,244.6
XS GIS Cut Line= 3
     2007301.953      372885.397     2007537.502      372394.012
     2007638.802      372227.079
#Sta/Elev= 30
       0 2573.32    19.8 2569.41    39.6 2566.16    69.4  2562.1    99.1 2557.72
   138.7 2551.44   178.3 2544.66     218  2539.4   247.7 2534.45   287.3    2530
   336.9 2522.92   356.7 2520.47   366.6  2519.6   396.3 2518.03     426 2515.62
   455.8 2512.61   525.1 2504.58     535  2503.7   540.7 2503.68   544.9 2503.67
   554.7 2505.39   555.7 2505.74   574.2  2512.6     584    2516   593.7 2518.99
   603.5  2521.5   613.3 2523.59     623 2525.43   642.6 2528.44   740.2 2541.14
#Mann= 3 , 0 , 0
       0      .1       0   540.7    .045       0   555.7      .1       0
Bank Sta=540.7,555.7
XS Rating Curve= 0 ,0
Exp/Cntr=0.3,0.1

Type RM Length L Ch R = 1 ,13539.5 ,300.5,304.9,309.3
XS GIS Cut Line= 2
     2007329.928      372917.732     2008116.164      372158.717
#Sta/Elev= 30
       0 2579.14    29.8 2571.32    79.5 2561.62   139.1 2558.97     159 2557.48
   178.8 2555.23   218.6 2548.65   288.1 2543.01     308 2540.72   407.3    2515
   437.1 2508.12   536.5 2498.37   538.7 2498.41   546.4 2498.54   553.7 2499.56
   596.1 2510.05   665.6 2529.24   705.4 2542.23     765 2564.19   784.8 2572.32
   844.5 2602.37   854.4 2607.07   864.3 2610.18   874.3 2609.74   894.1 2604.87
   904.1 2604.19     914 2605.06   963.7 2614.26  1003.4 2619.99  1092.8  2646.9
#Mann= 3 , 0 , 0
       0      .1       0   538.7    .045       0   553.7      .1       0
Bank Sta=538.7,553.7
XS Rating Curve= 0 ,0
Exp/Cntr=0.3,0.1

Type RM Length L Ch R = 1 ,13234.5 ,432.3,400.3,368.4
XS GIS Cut Line= 4
     2007761.543       373393.45     2007786.533      372857.841
     2007948.103      372753.817     2008073.364      372484.638
#Sta/Elev= 30
       0  2507.7    29.8  2510.6    89.4 2517.82   129.1 2523.72   178.7 2531.89
   198.6 2534.45   218.4 2536.42   248.2 2537.64     288 2537.32   307.8 2537.77
   367.4 2541.62   387.2 2541.79     417 2539.76   466.7 2534.74   536.2 2524.83
   574.6 2515.18   651.5 2497.68   670.7 2492.53   679.5 2491.33   680.3 2491.22
   689.9 2491.49   694.5 2492.28   748.2    2504   807.5 2518.52   886.7 2536.74
   906.5 2542.12   936.2 2552.09   965.9  2564.1   985.7 2573.95  1025.2 2597.19
#Mann= 3 , 0 , 0
       0      .1       0   679.5    .045       0   694.5      .1       0
Bank Sta=679.5,694.5
XS Rating Curve= 0 ,0
Exp/Cntr=0.3,0.1

Type RM Length L Ch R = 1 ,12833.9 ,292.6,293.9,295.1
XS GIS Cut Line= 3
     2008338.545       373294.84     2008133.436       372802.79
     2008136.661      372641.215
#Sta/Elev= 30
       0 2566.18    19.7 2560.47    29.6 2558.37    39.5 2556.59     158 2538.03
   187.6 2533.18   207.3 2529.63   227.1 2525.24   256.7 2517.31   266.5 2514.98
     306 2506.95   335.6 2501.62     385 2493.94   404.8 2490.42   414.6 2489.14
   416.9 2489.09   424.5 2488.93   431.9  2489.3   444.2 2490.26     464 2492.19
   513.3 2497.65   542.6 2501.41   561.6 2504.45   571.1 2506.25   590.1 2510.35
   609.1 2514.84   628.2 2519.66   647.2 2524.97   675.7 2533.67   694.7 2538.92
#Mann= 3 , 0 , 0
       0      .1       0   416.9    .045       0   431.9      .1       0
Bank Sta=416.9,431.9
XS Rating Curve= 0 ,0
Exp/Cntr=0.3,0.1

Type RM Length L Ch R = 1 ,12539.8 ,479.3,474,468.7
XS GIS Cut Line= 2
     2008510.447         373015.     2008326.552      372487.303
#Sta/Elev= 30
       0 2532.63    29.9 2526.78    59.9 2521.47   119.8 2511.78   149.7 2506.63
   159.7 2505.06   179.6 2502.46   189.6 2500.85   229.5 2494.05   249.5 2490.34
   256.7  2489.5   259.4 2489.18   269.4 2489.76   271.7 2490.45   279.4 2492.74
   289.4 2496.98   299.4  2500.6   319.3 2506.83   339.3 2512.33   369.2 2519.97
   429.1 2534.45   439.1 2537.24     469 2547.55     479 2551.43     489 2556.05
     499 2561.06   508.9  2566.4   518.9 2572.12   548.8 2590.18   558.8 2595.89
#Mann= 3 , 0 , 0
       0      .1       0   256.7    .045       0   271.7      .1       0
Bank Sta=256.7,271.7
XS Rating Curve= 0 ,0
Exp/Cntr=0.3,0.1

Type RM Length L Ch R = 1 ,12065.5 ,703.6,707.6,711
XS GIS Cut Line= 2
     2009076.122      372993.013     2008694.341      372389.359
#Sta/Elev= 30
       0 2588.44    29.8  2578.5    69.4 2561.93    79.4 2558.19    99.2 2551.91
     119 2547.04   148.8 2541.39   218.2 2527.04   317.4 2508.68     377 2500.14
   406.7 2497.16   446.4 2494.42   456.3 2492.12   476.2 2484.54   479.1  2484.1
   486.1 2483.03   494.1 2484.15     496 2484.41   505.9 2489.82   515.8 2496.18
   525.8 2501.38   535.7 2505.07   545.6 2507.33   555.5 2508.93     615 2515.94
   644.8 2520.88   664.6 2525.58   684.5 2531.24   704.3 2538.62   714.2 2542.97
#Mann= 3 , 0 , 0
       0      .1       0   479.1    .045       0   494.1      .1       0
Bank Sta=479.1,494.1
XS Rating Curve= 0 ,0
Exp/Cntr=0.3,0.1

Type RM Length L Ch R = 1 ,11357.7 ,294.3,298.4,303
XS GIS Cut Line= 3
      2009481.89      372731.163     2009286.225      372223.817
     2009176.065      371971.599
#Sta/Elev= 30
       0 2594.15    19.8 2589.34    39.6 2583.14    69.2 2571.95   108.8 2555.91
   118.6 2552.63   128.5 2550.23   168.1 2542.08   187.8 2538.31   237.3 2529.67
   276.8 2521.78   296.6 2517.22   306.5 2514.62   326.3 2508.73     346 2503.96
   365.8 2500.72   395.5    2497   454.8 2490.83   504.2 2486.43   547.5 2480.06
   553.6 2479.36   562.5 2479.79   573.3 2482.28   592.9 2489.91   651.9 2509.26
   671.6 2516.25   691.2 2524.03   730.5 2538.81   779.7  2559.4     819 2574.77
#Mann= 3 , 0 , 0
       0      .1       0   547.5    .045       0   562.5      .1       0
Bank Sta=547.5,562.5
XS Rating Curve= 0 ,0
Exp/Cntr=0.3,0.1

Type RM Length L Ch R = 1 ,11059.3 ,400.3,403.9,407.6
XS GIS Cut Line= 2
      2009673.11      372764.982     2009436.426      371651.736
#Sta/Elev= 30
       0 2614.63    79.9 2597.32    99.8 2592.04   199.7 2553.49   369.4 2514.95
   479.2 2492.46   489.2 2489.21   509.2 2479.34   519.2 2477.56   529.3 2478.29
   544.3 2479.94     639  2485.3   658.9 2487.19   668.9 2489.16   718.8 2504.02
   778.7  2523.9   798.7  2531.5   828.6 2544.04   858.6 2557.61   878.6 2567.56
   908.5 2584.02   918.5  2588.6   928.5 2590.72   958.4 2588.37   988.4 2588.86
   998.4  2590.6  1028.3  2599.1  1068.2  2604.8  1118.2 2615.67  1138.1 2621.24
#Mann= 3 , 0 , 0
       0      .1       0   529.3    .045       0   544.3      .1       0
Bank Sta=529.3,544.3
XS Rating Curve= 0 ,0
Exp/Cntr=0.3,0.1

Type RM Length L Ch R = 1 ,10655.1 ,492.2,488.5,484.9
XS GIS Cut Line= 3
     2009869.667      372565.258      2009926.93      372241.606
      2009899.65      371785.705
#Sta/Elev= 30
       0 2551.42      10 2547.77    19.9 2544.78    39.8 2539.84    49.8  2537.8
    79.7 2532.55    99.6 2528.59   169.3 2513.22   209.2 2505.21     259  2494.9
   278.9 2490.46   308.8 2482.95   318.7 2481.04   328.7 2479.92   368.4 2476.99
   421.4 2472.01   436.4 2470.88   437.9 2470.79   447.8 2470.89   457.8 2472.04
   487.5  2478.6   537.2 2488.85     557 2493.28   586.8 2499.28   596.8 2501.51
   616.6 2506.37   676.2 2521.88   725.8  2535.1   755.6 2543.72   785.4 2553.29
#Mann= 3 , 0 , 0
       0      .1       0   421.4    .045       0   436.4      .1       0
Bank Sta=421.4,436.4
XS Rating Curve= 0 ,0
Exp/Cntr=0.3,0.1

Type RM Length L Ch R = 1 ,10165.7 ,413,430.3,447.7
XS GIS Cut Line= 4
     2010388.036      372424.006     2010181.719       371536.14
     2009848.725      370963.362     2009687.843       370285.83
#Sta/Elev= 30
       0 2521.42    70.1 2510.12   200.3 2482.43   240.4 2475.59   270.4 2472.52
   350.6 2471.54   384.7 2468.55   399.7 2466.48   400.7 2466.35   410.7 2468.09
   430.7 2479.48   440.7 2482.96   510.8 2501.86   550.9 2509.93     611 2511.01
   771.3 2520.59   821.4  2518.5   911.5 2507.29  1089.5 2492.87  1119.2 2492.28
  1198.3 2495.17  1307.1 2485.83  1356.5 2483.04  1445.5 2484.06  1485.1 2486.44
  1613.9 2498.05  1713.3 2510.09  1822.8 2515.34  1882.5 2515.27  2270.4 2500.45
#Mann= 3 , 0 , 0
       0      .1       0   384.7    .045       0   399.7      .1       0
Bank Sta=384.7,399.7
XS Rating Curve= 0 ,0
Exp/Cntr=0.3,0.1

Type RM Length L Ch R = 1 ,9735.1  ,401.9,408.8,417.1
XS GIS Cut Line= 5
     2010553.941      372393.357     2010815.608       371951.23
     2010614.523      371440.706      2010067.79      370643.746
     2009961.708      370275.397
#Sta/Elev= 30
       0 2523.76      79 2510.54   128.4 2493.37   217.4 2476.19   257.7 2464.04
   266.8 2463.84   272.7 2463.88   464.4 2481.14   603.5 2488.89   733.2 2489.58
   803.1 2486.16   922.8 2485.08   982.6 2493.76  1092.4 2506.77  1152.1 2517.85
  1221.9 2522.13  1341.4 2519.88  1490.9 2512.75  1510.8 2513.42  1560.6 2522.38
  1580.6 2523.46  1670.2 2515.59    1720 2513.09    1740 2514.23  1779.8  2521.8
  1809.7  2523.5  2028.9 2502.05  2284.5 2502.91  2372.9 2493.27  2412.2 2491.21
#Mann= 3 , 0 , 0
       0      .1       0   257.7    .045       0   272.7      .1       0
Bank Sta=257.7,272.7
XS Rating Curve= 0 ,0
Exp/Cntr=0.3,0.1

Type RM Length L Ch R = 1 ,9326.4  ,305.3,299.6,291.6
XS GIS Cut Line= 3
     2010580.771      372786.668     2011004.118      372410.973
     2011436.557      372070.498
#Sta/Elev= 30
       0 2609.22    49.6 2605.63    79.4 2602.54   109.2 2598.37   129.1 2594.14
   178.7 2578.67   228.4 2560.78     288 2544.18   317.8 2535.08   476.6 2474.89
   486.6 2472.07   506.4 2468.38   558.5 2462.41   573.5 2461.06     576 2460.94
     586 2461.37     596 2462.71     626 2468.19   676.1 2475.08   686.1 2477.03
   746.1  2493.1   836.2 2514.82   856.2 2520.82   886.2 2531.59   966.3 2564.06
   996.3 2575.34  1016.3 2581.93  1036.3 2587.65  1066.4 2593.75  1116.4 2609.78
#Mann= 3 , 0 , 0
       0      .1       0   558.5    .045       0   573.5      .1       0
Bank Sta=558.5,573.5
XS Rating Curve= 0 ,0
Exp/Cntr=0.3,0.1

Type RM Length L Ch R = 1 ,9026.4  ,306.7,300,292.1
XS GIS Cut Line= 3
     2010892.141      373083.066     2011190.447       372635.61
     2011498.573      372129.415
#Sta/Elev= 30
       0 2633.52    19.9 2628.15    39.8 2621.63   258.9 2544.72   278.8 2538.44
   328.6  2523.9   368.5 2511.31   398.4 2501.48   497.9 2466.28   517.9 2458.63
   527.8 2455.42   530.3 2455.21   537.8 2454.58   545.3 2454.86   685.9 2468.27
   695.8 2469.35   705.7 2471.05   715.6 2473.96   725.4 2477.55   774.8 2497.08
   784.7 2500.62   873.6 2525.54   913.1 2537.48   942.7 2547.17   962.5 2554.34
   972.4 2558.32   992.1 2567.15  1021.7 2581.31  1031.6 2585.45  1130.4 2614.42
#Mann= 3 , 0 , 0
       0      .1       0   530.3    .045       0   545.3      .1       0
Bank Sta=530.3,545.3
XS Rating Curve= 0 ,0
Exp/Cntr=0.3,0.1

Type RM Length L Ch R = 1 ,8726.4  ,292.3,300,310.3
XS GIS Cut Line= 3
     2011324.427      373246.552     2011473.801      372689.105
     2011578.275      372157.721
#Sta/Elev= 30
       0 2604.82    39.8 2595.43    79.6 2584.11    99.5 2577.67   119.4 2569.83
   139.3 2563.11   218.9 2539.78   467.7 2471.32   487.6 2467.12   569.6 2453.67
   577.1 2452.91   584.6 2453.02   596.8 2454.18   626.4 2459.13     646 2463.39
   665.7 2468.92   695.3 2479.97   744.5 2501.91     774 2513.65     843 2535.42
   961.1  2576.9   980.8 2580.73   990.7 2584.24  1010.4 2593.42  1020.2 2596.93
  1069.4 2610.69  1089.1 2615.67    1099 2617.42  1108.8  2617.9  1118.7 2617.08
#Mann= 3 , 0 , 0
       0      .1       0   569.6    .045       0   584.6      .1       0
Bank Sta=569.6,584.6
XS Rating Curve= 0 ,0
Exp/Cntr=0.3,0.1

Type RM Length L Ch R = 1 ,8426.4  ,407.3,419.7,431.7
XS GIS Cut Line= 3
     2011402.706      373284.397     2011740.278       372818.42
     2012066.445      372387.037
#Sta/Elev= 30
       0 2594.16    79.4 2573.72   238.1  2528.8   337.3 2502.16   367.1 2492.59
   406.8  2478.3   436.5 2464.63   446.4 2460.96   456.4  2459.1     496  2456.5
   565.5 2450.12   567.9 2450.29   575.4 2450.84   582.9 2452.83   605.4 2461.84
   625.5 2468.61   655.5 2477.77   705.6 2491.02   725.6 2494.76   785.7 2502.69
   885.9  2522.1   905.9 2526.95   935.9  2535.9     986 2556.72     996 2559.59
    1006 2561.05  1036.1 2560.67  1066.1 2562.01  1096.2 2567.79  1116.2  2572.7
#Mann= 3 , 0 , 0
       0      .1       0   567.9    .045       0   582.9      .1       0
Bank Sta=567.9,582.9
XS Rating Curve= 0 ,0
Exp/Cntr=0.3,0.1

Type RM Length L Ch R = 1 ,8006.6  ,276.6,279.9,283.2
XS GIS Cut Line= 3
      2011475.63      373368.791     2012016.837      373141.885
      2012236.31      373003.007
#Sta/Elev= 30
       0 2586.73    19.9 2579.06    29.8  2575.7   139.2 2540.02     189 2524.23
   278.5 2497.24   308.3 2486.84     378 2460.09   387.9 2456.46   397.9 2453.35
   407.8 2451.64   417.8 2451.16   477.4 2451.86   507.3 2451.34   527.2  2450.1
   537.1 2448.86   556.3 2445.06     567 2444.57   571.3 2445.42   576.9 2446.52
   596.8 2453.44   606.8 2455.87   686.7 2468.49   696.7  2470.5   716.7 2475.71
   756.7 2485.23   776.6 2491.37   796.6 2498.42   816.6 2506.36   846.6 2519.46
#Mann= 3 , 0 , 0
       0      .1       0   556.3    .045       0   571.3      .1       0
Bank Sta=556.3,571.3
XS Rating Curve= 0 ,0
Exp/Cntr=0.3,0.1

Type RM Length L Ch R = 1 ,7726.8  ,209.2,201.1,193.1
XS GIS Cut Line= 3
     2011538.248       373543.33      2012148.36      373392.783
     2012300.273      373318.826
#Sta/Elev= 30
       0  2582.5    29.9 2571.95    69.8 2559.34    79.8 2555.91   109.7 2544.71
   159.6 2526.54   199.5 2512.57   229.4 2503.07   259.3 2494.42   289.3  2486.9
   349.1 2473.64     399 2461.62     409 2459.52   418.9 2457.98   448.9 2454.12
   468.8 2451.03   488.8 2447.56   518.7 2441.15   529.4 2439.78   538.6 2439.57
   544.4 2439.94   558.6 2441.29   608.5 2446.88   668.2 2454.52     688 2457.57
     698 2459.85   767.6 2480.93   777.5  2484.2   787.4 2487.89   797.4    2492
#Mann= 3 , 0 , 0
       0      .1       0   529.4    .045       0   544.4      .1       0
Bank Sta=529.4,544.4
XS Rating Curve= 0 ,0
Exp/Cntr=0.3,0.1

Type RM Length L Ch R = 1 ,7525.6  ,364.9,354.4,343.7
XS GIS Cut Line= 3
     2011684.626      373756.575     2012116.378      373610.658
       2012428.2      373394.782
#Sta/Elev= 30
       0 2563.77    29.7 2552.67    39.6 2549.53   178.3  2510.8   198.2 2504.71
   227.9 2494.66   336.8 2456.79   346.8 2453.58   356.7 2450.96   366.6 2449.14
   376.5 2447.85     426 2442.22   455.7 2440.47   485.7 2438.27   489.8 2438.28
   495.7  2438.3   504.8  2439.1   535.6 2443.05   575.5 2447.15   595.5 2449.51
   615.4 2452.16   625.4 2454.02   635.4 2456.66   655.4 2462.63   675.3 2468.19
   725.2 2481.47   745.2 2487.37   765.1 2494.01   775.1 2497.61     835 2521.18
#Mann= 3 , 0 , 0
       0      .1       0   489.8    .045       0   504.8      .1       0
Bank Sta=489.8,504.8
XS Rating Curve= 0 ,0
Exp/Cntr=0.3,0.1

Type RM Length L Ch R = 1 ,7171.1  ,260.5,252.8,245.3
XS GIS Cut Line= 3
     2012205.661       374148.35     2012416.206      373777.896
     2012682.536      373344.483
#Sta/Elev= 30
       0  2508.4    39.6 2494.05    79.3 2476.73    99.1  2469.3   128.8 2459.34
   158.6 2450.85   168.5 2448.58   178.4 2447.27   267.6 2441.46   307.2 2435.14
   316.9 2434.76   331.9 2434.99   426.1 2438.73   436.1 2439.71     446 2442.12
     476 2454.32     486 2457.58   615.6 2493.96   715.4 2523.77   735.3 2528.47
   765.2 2534.17   775.2 2535.63   795.2  2536.7   805.1 2538.07   815.1 2543.31
   825.1 2550.95   835.1  2557.1     845 2561.93   904.9 2589.43   934.8 2600.99
#Mann= 3 , 0 , 0
       0      .1       0   316.9    .045       0   331.9      .1       0
Bank Sta=316.9,331.9
XS Rating Curve= 0 ,0
Exp/Cntr=0.3,0.1

Type RM Length L Ch R = 1 ,6918.3  ,526.9,540.6,554.2
XS GIS Cut Line= 3
     2012376.229      374500.148     2012565.454       374049.74
     2012637.413      373604.662
#Sta/Elev= 30
       0 2608.47    19.9  2603.7    49.8 2594.56    59.8 2590.22    69.8 2584.64
   119.6 2555.28   139.6 2545.74   169.5 2534.88   219.4 2519.34   239.3 2512.26
   269.2 2500.21     339  2469.9   388.8 2450.81   398.8  2448.2   408.8 2446.74
   478.6 2440.62   488.5 2439.02   508.1 2434.23     518 2432.64   527.8 2432.24
   528.7 2432.26   543.7 2432.56     665 2433.14   684.6 2434.27   694.4 2435.92
   733.6 2444.22     812 2458.66   831.6 2463.02   851.2 2469.28   939.4 2501.33
#Mann= 3 , 0 , 0
       0      .1       0   528.7    .045       0   543.7      .1       0
Bank Sta=528.7,543.7
XS Rating Curve= 0 ,0
Exp/Cntr=0.3,0.1

Type RM Length L Ch R = 1 ,6377.2  ,511.4,500.3,489.2
XS GIS Cut Line= 4
     2012810.647      374468.167     2012938.574      374180.332
     2013065.343      374048.526     2013087.821      373876.506
#Sta/Elev= 30
       0 2512.83    19.7 2506.35    29.5 2501.14    49.2 2488.98    68.9 2479.21
    78.8 2475.72   118.1 2464.07   167.3 2447.89     187 2442.32   206.7 2437.56
   226.4 2434.28   255.9 2431.93   334.2 2429.69   353.5 2428.58   382.4 2424.68
   420.9 2418.58   425.6 2418.27   430.5 2417.94   440.6 2418.21   459.4 2419.82
     469 2421.43   488.2 2425.75   497.9 2429.31   517.1 2438.19   526.8  2441.1
   536.4 2442.59     575 2445.62   594.2 2447.93   632.8 2453.96   671.3 2461.69
#Mann= 3 , 0 , 0
       0      .1       0   425.6    .045       0   440.6      .1       0
Bank Sta=425.6,440.6
XS Rating Curve= 0 ,0
Exp/Cntr=0.3,0.1

Type RM Length L Ch R = 1 ,5877    ,451,450.8,450.5
XS GIS Cut Line= 2
      2013351.67      374692.038      2013538.23      374025.754
#Sta/Elev= 30
       0  2464.7    29.6 2458.71    59.3 2453.28    69.2 2451.92    79.1 2450.95
    98.8 2447.76   118.6 2444.89   187.8 2437.86   316.3 2426.52   326.2 2425.37
   336.1 2423.22     346 2419.58   355.8 2414.79   365.7 2410.25   375.6 2407.97
   384.8 2407.98   399.8 2409.57   415.2 2411.24     425 2412.05   454.7 2413.92
   484.3 2415.02   543.6 2415.72   563.4 2416.15   573.3 2416.62   583.2 2418.02
   593.1 2420.74     603 2424.08   642.5 2437.92   672.1 2448.73   691.9 2455.66
#Mann= 3 , 0 , 0
       0      .1       0   384.8    .045       0   399.8      .1       0
Bank Sta=384.8,399.8
XS Rating Curve= 0 ,0
Exp/Cntr=0.3,0.1

Type RM Length L Ch R = 1 ,5426.2  ,645.8,641.1,636.7
XS GIS Cut Line= 3
     2013702.802      374838.177     2013853.231      374529.956
     2013966.651      374106.596
#Sta/Elev= 30
       0 2490.07    68.6 2471.81   107.8 2460.59     147 2448.75   166.6 2443.01
   176.4 2440.21   186.2 2437.66   205.8 2432.94   225.4 2428.73   264.6 2421.68
   284.2 2418.49   313.6 2414.11   372.8 2405.83   382.8 2404.69   392.8 2404.06
   422.7 2403.19   442.6 2402.42     541 2397.68     556 2396.89   572.1 2396.26
     582 2396.55     592 2398.31     602 2401.44   611.9 2405.08   621.9 2408.52
   671.7 2424.65   681.6 2428.23   711.5 2439.74   751.4 2454.39   781.3 2465.78
#Mann= 3 , 0 , 0
       0      .1       0     541    .045       0     556      .1       0
Bank Sta=541,556
XS Rating Curve= 0 ,0
Exp/Cntr=0.3,0.1

Type RM Length L Ch R = 1 ,4784.9  ,550.3,572.7,594.8
XS GIS Cut Line= 4
     2014313.185      374925.913     2014428.773      374696.673
     2014448.335      374454.107      2014415.08      374338.693
#Sta/Elev= 30
       0 2446.39    19.8 2444.03    29.6 2443.27    49.4 2442.39    59.2 2441.07
    69.1 2438.33      79 2434.93   118.5 2420.75   128.4 2417.61   138.2 2415.45
     158 2412.45   167.9  2410.7   197.5 2404.19   217.2 2400.33     237 2396.75
   246.9 2394.71   266.5 2389.22   276.2 2388.07   285.9 2387.95   300.3 2388.16
   315.3 2388.38   500.1 2389.96   510.1 2390.24   520.1 2391.26   530.1 2393.63
   550.1 2399.79   560.1 2402.67   590.2 2410.61   600.2  2413.7   620.2 2421.42
#Mann= 3 , 0 , 0
       0      .1       0   300.3    .045       0   315.3      .1       0
Bank Sta=300.3,315.3
XS Rating Curve= 0 ,0
Exp/Cntr=0.3,0.1

Type RM Length L Ch R = 1 ,4212.4  ,306.7,305.3,304
XS GIS Cut Line= 5
      2014563.75       375005.75     2014706.551      374851.211
     2014857.176      374718.191     2014949.117      374663.418
     2015199.507      374495.187
#Sta/Elev= 30
       0 2414.36    38.3 2409.89      67 2407.08    86.1 2405.01   114.8 2401.48
   172.2 2393.83   181.7 2392.69   200.8 2390.81     220 2389.39   239.1 2388.21
   267.8  2387.1     354 2383.15   483.9 2376.42   489.2 2376.25   498.9 2376.46
   508.7 2377.62   528.1 2381.36   537.8 2382.93   547.6 2384.17   557.3  2384.7
   576.8 2385.05   586.5 2385.46     606  2386.9   615.7  2387.8   644.9 2391.07
   703.3 2399.02   742.2 2403.92   751.9 2405.39   761.7 2407.29     820 2419.56
#Mann= 3 , 0 , 0
       0      .1       0   483.9    .045       0   498.9      .1       0
Bank Sta=483.9,498.9
XS Rating Curve= 0 ,0
Exp/Cntr=0.3,0.1

Type RM Length L Ch R = 1 ,3906.8  ,280.8,280.3,279.6
XS GIS Cut Line= 3
     2014841.527      375195.499     2014999.977      374988.144
      2015368.28      374742.436
#Sta/Elev= 30
       0 2413.26    48.3 2405.39      58 2403.92    77.3 2401.29   106.3  2397.7
   154.6 2392.35     203 2387.55   212.6 2386.34   251.3  2380.8     261 2379.55
   280.6 2375.84   290.5 2374.77   300.3 2374.53   349.5 2374.01   413.2 2373.61
   418.4 2373.59   428.2 2374.23   438.1  2376.4   457.7 2382.76   467.6  2385.3
   477.4 2387.39   487.2 2389.01   506.9 2391.87   546.3  2397.1   575.8 2401.25
   595.5 2404.43   605.3 2406.41   615.2 2408.74   644.7 2416.08   703.7 2431.51
#Mann= 3 , 0 , 0
       0      .1       0   413.2    .045       0   428.2      .1       0
Bank Sta=413.2,428.2
XS Rating Curve= 0 ,0
Exp/Cntr=0.3,0.1

Type RM Length L Ch R = 1 ,3626.4  ,301.3,299.9,299.3
XS GIS Cut Line= 3
     2015070.018      375265.931      2015224.15      375157.908
     2015391.833      375038.062
#Sta/Elev= 30
       0 2412.19     9.9 2410.45    19.8 2408.47    29.7 2406.21    39.6  2403.6
    49.5 2400.36    59.4  2396.4    79.2 2387.67    89.2 2383.49    99.1  2379.8
     109  2377.2   118.9 2375.71   128.8 2374.96   148.6 2373.63   158.5 2372.68
   168.4 2371.47   178.3 2370.61   180.7 2370.62   188.2 2370.64   195.7 2371.66
     198 2371.97   207.8 2373.67   217.7  2375.1   276.6  2382.4   296.2 2384.98
   325.6  2389.2   335.4 2390.67   355.1 2393.91   384.5 2399.35   394.3 2401.36
#Mann= 3 , 0 , 0
       0      .1       0   180.7    .045       0   195.7      .1       0
Bank Sta=180.7,195.7
XS Rating Curve= 0 ,0
Exp/Cntr=0.3,0.1

Type RM Length L Ch R = 1 ,3326.4  ,304.5,300.1,295.4
XS GIS Cut Line= 3
        2015015.      375693.245     2015442.272      375349.542
     2015882.651      375019.357
#Sta/Elev= 30
       0  2517.4   159.5 2461.16   219.3 2441.36   289.1 2419.87   309.1 2413.36
   388.8 2384.59   398.8 2381.26   408.8 2378.64   418.7 2377.43   458.6 2374.87
   498.5  2371.3   528.4 2367.91   540.9 2366.94   548.4 2366.89   555.9 2367.92
   578.4    2373   648.4 2386.52   758.5 2409.25   798.5 2417.93   838.6  2425.7
   898.6  2438.2   908.6 2440.73   918.6 2443.98   948.7 2454.88   968.7 2460.85
   998.7 2468.24  1048.7 2478.87  1068.8 2483.61  1078.8 2486.68  1098.8 2494.09
#Mann= 3 , 0 , 0
       0      .1       0   540.9    .045       0   555.9      .1       0
Bank Sta=540.9,555.9
XS Rating Curve= 0 ,0
Exp/Cntr=0.3,0.1

Type RM Length L Ch R = 1 ,3026.4  ,294.4,300,304
XS GIS Cut Line= 3
     2015311.887      375966.407     2015663.142      375548.189
      2016023.26      375137.822
#Sta/Elev= 30
       0 2542.34   129.1 2491.42   258.2 2439.71   268.1 2436.31     278 2434.23
   297.9 2430.93   307.8 2427.48   317.8 2423.33   357.5 2406.15   377.3 2399.18
   407.1 2389.63     427 2383.67   456.8 2376.32   466.7 2374.39   476.6 2373.13
   538.7 2366.11   546.2  2365.8   553.7 2366.65   556.1 2366.92     566 2369.31
   615.6 2382.74   645.4 2390.17   665.3 2394.17   754.6 2410.72   873.7  2440.1
   903.5 2446.46   933.3 2451.82   953.2 2455.84  1042.5 2477.48  1092.1  2491.3
#Mann= 3 , 0 , 0
       0      .1       0   538.7    .045       0   553.7      .1       0
Bank Sta=538.7,553.7
XS Rating Curve= 0 ,0
Exp/Cntr=0.3,0.1

Type RM Length L Ch R = 1 ,2726.4  ,305.5,300,295.5
XS GIS Cut Line= 3
     2015414.879      376091.352     2015858.324      375773.584
        2016287.      375431.504
#Sta/Elev= 30
       0 2535.05    39.7 2515.96    59.5  2507.6    69.4 2504.44    99.2  2496.7
     129 2485.66     248  2445.1   297.6 2426.95   307.5 2423.96   317.4 2422.39
   337.2 2421.63   347.2 2420.43   357.1 2417.31   406.7 2396.74   466.2 2377.86
   476.1  2375.7     496 2372.92     538 2365.41   545.6 2364.61     553 2364.61
   605.4  2370.9   675.2 2373.94   705.1 2376.26     735 2380.52   764.9 2386.14
   784.9 2390.73   804.8 2396.13   884.6 2421.01   954.4 2439.87    1094 2480.57
#Mann= 3 , 0 , 0
       0      .1       0     538    .045       0     553      .1       0
Bank Sta=538,553
XS Rating Curve= 0 ,0
Exp/Cntr=0.3,0.1

Type RM Length L Ch R = 1 ,2426.4  ,290.6,292.7,295
XS GIS Cut Line= 3
     2015725.122      376390.906     2016078.992      375975.108
     2016429.608      375556.531
#Sta/Elev= 30
       0 2529.61    99.3 2494.31   198.5 2454.74   228.3 2446.29     278  2435.3
   337.5 2418.74   347.4 2416.96   357.4 2415.76   367.3  2413.8   377.2 2410.15
   416.9 2392.54   436.8 2384.68   486.4 2370.58   526.1 2361.28   536.1 2360.26
   538.5 2360.37     546 2360.73   553.5 2361.71   595.6 2366.86   625.4 2369.78
   694.9 2375.84   734.6 2378.27   754.5 2380.88   784.3 2386.99   804.1 2392.31
     814 2395.45   883.5 2420.79   913.3  2430.9  1052.3 2474.04    1092 2485.85
#Mann= 3 , 0 , 0
       0      .1       0   538.5    .045       0   553.5      .1       0
Bank Sta=538.5,553.5
XS Rating Curve= 0 ,0
Exp/Cntr=0.3,0.1

Type RM Length L Ch R = 1 ,2133.7  ,320.3,319.7,319.2
XS GIS Cut Line= 2
      2015910.76      376545.361     2016655.775      375819.614
#Sta/Elev= 30
       0 2512.85     100  2480.9     150 2464.41     210 2443.86     230  2437.6
     280 2422.71     290  2420.2     310 2417.66     320 2414.42     350 2399.66
     360 2395.03     370 2390.99     430 2372.47     450 2366.87     500 2356.84
     520 2352.18     530 2350.31     540 2349.61   540.8 2349.65     550 2350.05
   555.8 2350.88     610 2358.87     650 2365.41     670 2369.35     710 2378.48
     760 2388.72   830.1 2404.35   950.1 2429.54   980.1 2437.02  1040.1 2453.83
#Mann= 3 , 0 , 0
       0      .1       0   540.8    .045       0   555.8      .1       0
Bank Sta=540.8,555.8
XS Rating Curve= 0 ,0
Exp/Cntr=0.3,0.1

Type RM Length L Ch R = 1 ,1813.8  ,293.3,283.3,273.3
XS GIS Cut Line= 2
     2016165.389      376744.417     2016883.379       376024.47
#Sta/Elev= 30
       0 2471.72    29.9 2461.37    59.8 2451.56   139.6  2427.4     299 2377.09
   348.9 2362.32   388.8  2351.7   398.7 2349.68   418.7 2347.02   446.2 2345.03
   458.6 2344.38   461.2 2344.41   468.5  2344.5   478.5 2345.67   498.4    2349
   558.2    2358   598.1  2364.8   667.9 2381.19   757.6 2403.87   777.5 2409.33
   807.4 2418.42   837.3 2426.27   857.3 2430.06   867.2 2431.26   907.1 2433.96
   927.1 2436.76     947 2441.02   966.9  2446.2   986.9 2452.07  1016.8 2461.57
#Mann= 3 , 0 , 0
       0      .1       0   446.2    .045       0   461.2      .1       0
Bank Sta=446.2,461.2
XS Rating Curve= 0 ,0
Exp/Cntr=0.3,0.1

Type RM Length L Ch R = 1 ,1530.5  ,405.2,414,422.7
XS GIS Cut Line= 2
     2016505.377      377133.824     2016864.555      376074.928
#Sta/Elev= 30
       0 2510.41      30 2499.95    69.9 2485.29    79.9 2482.01    99.8 2477.32
   109.8 2474.47   179.7 2451.45   259.6 2424.12   319.5  2402.9   349.4 2392.87
   379.4 2381.25   399.3 2374.31   429.3 2366.35   469.2  2357.1   529.1 2345.66
   539.1 2344.22   549.1 2343.89   554.2 2344.16   569.2  2345.3   698.8 2354.55
   728.8 2357.62   758.8 2361.89   838.6 2378.47   878.6 2388.37   918.5 2397.51
   968.4 2410.03  1048.3 2425.81  1078.2 2432.12  1098.2 2437.78  1118.2 2444.24
#Mann= 3 , 0 , 0
       0      .1       0   554.2    .045       0   569.2      .1       0
Bank Sta=554.2,569.2
XS Rating Curve= 0 ,0
Exp/Cntr=0.3,0.1

Type RM Length L Ch R = 1 ,1116.5  ,421.7,413.4,405
XS GIS Cut Line= 3
     2016693.087      377141.522     2017071.302      376725.304
     2017196.798      376437.926
#Sta/Elev= 30
       0 2481.52    69.1 2454.66   108.5 2441.16   177.6 2419.72   305.9 2382.91
   315.7 2379.82   394.7 2352.87   404.5 2350.11   414.4  2347.9   434.1 2344.35
   463.7 2340.28   483.5 2336.87   493.3 2335.83   503.2 2335.79   511.1    2336
   526.1 2336.46   542.7 2337.51   572.2 2340.47   611.4 2343.45   640.8 2344.94
   689.8 2346.77   719.2 2348.38   738.8 2350.11   758.4 2352.62     778 2356.16
   797.6 2360.81   817.2 2365.96     827 2369.14   856.4 2380.01     876 2386.32
#Mann= 3 , 0 , 0
       0      .1       0   511.1    .045       0   526.1      .1       0
Bank Sta=511.1,526.1
XS Rating Curve= 0 ,0
Exp/Cntr=0.3,0.1

Type RM Length L Ch R = 1 ,703.1   ,414.9,424.3,433.7
XS GIS Cut Line= 3
      2017151.49      377216.146     2017367.367      377021.591
     2017574.851      376466.755
#Sta/Elev= 30
       0 2409.59    48.4 2396.13   135.6 2374.06   174.4 2363.67   213.1 2352.78
   242.2 2342.88   251.9 2340.12   271.2 2335.48   300.5 2329.51   310.4 2327.86
   320.2  2327.3   329.3 2327.48   344.3    2328     419 2329.97   448.6 2331.19
   468.3 2332.82   507.8  2337.2   537.4 2340.94   586.8 2349.25     646 2358.29
   685.5 2365.05   695.4 2366.38   705.3 2367.26   715.1 2367.67   734.9 2367.66
   784.2 2366.46   833.6 2364.91   843.5  2364.9   853.4 2365.23     883 2367.08
#Mann= 3 , 0 , 0
       0      .1       0   329.3    .045       0   344.3      .1       0
Bank Sta=329.3,344.3
XS Rating Curve= 0 ,0
Exp/Cntr=0.3,0.1

Type RM Length L Ch R = 1 ,278.8   ,257.4,252.4,248
XS GIS Cut Line= 3
     2017439.325      377298.765     2017713.835      377216.146
     2018027.624      376892.967
#Sta/Elev= 30
       0 2349.93    19.8 2345.26    39.5 2341.14    49.4 2339.27    59.3 2337.54
    69.2 2335.98    79.1 2334.58      89 2333.36    98.8 2332.43   108.7 2331.75
   138.4 2329.99   207.6 2325.54   276.8 2320.92   296.7 2319.32   306.7 2318.64
   315.6 2318.58   316.7 2318.57   330.6 2319.03   376.8 2321.16   396.8 2322.26
   416.8 2323.44   506.9  2329.2   556.9 2331.71     577 2332.43     587 2332.69
     607  2332.9     637 2332.85   667.1 2332.56   697.1 2331.63   737.1 2329.78
#Mann= 3 , 0 , 0
       0      .1       0   315.6    .045       0   330.6      .1       0
Bank Sta=315.6,330.6
XS Rating Curve= 0 ,0
Exp/Cntr=0.3,0.1
